--- MLLSTNCK.prj (project) ---

Proj Title=MLLSTNCK
Current Plan=p01
Default Exp/Contr=0,0
English Units
Geom File=g01
Flow File=f01
Plan File=p01
Background Map Layer=Inundation Boundary (01pct Value_0)
BEGIN DESCRIPTION:
----------MODEL BY WOOD PLC 2021----------
Stream Name: Millstone Creek
Flood Zone: Enhanced Approximate
Pocahontas County, WV
HEC-RAS Version: RAS 6.1.0
Vertical Datum: NAVD88
Projection: NAD 1983 StatePlane West Virginia S FIPS 4702 (US Feet)
Terrain: 1-meter LIDAR (FEMA Region III 3DEP collected 2016-2018)
Land Use: 2019 NLCD
Hydrologic Method:
WV SIR2010-5033 regression equations
Model Notes:
Heavy Karst area, spotty floodplain and sinkholes throughout the reach
END DESCRIPTION:
DSS File=dss
DSS Export Rating Curves= 0
DSS Export Rating Curve Sorted= 0
DSS Export Volume Flow Curves= 0
DXF OffsetX= 0
DXF OffsetY= 0
DXF ScaleX= 0
DXF ScaleY= 0

--- MLLSTNCK.p01 (plan) ---

Plan Title=Floodplain
Program Version=6.10
Short Identifier=Floodplain
Geom File=g01
Flow File=f01
Subcritical Flow
K Sum by GR= 0
Std Step Tol= 0.01
Critical Tol= 0.01
Num of Std Step Trials= 20
Max Error Tol= 0.3
Flow Tol Ratio= 0.001
Split Flow NTrial= 30
Split Flow Tol= 0.02
Split Flow Ratio= 0.02
Log Output Level= 0
Friction Slope Method= 1
Unsteady Friction Slope Method= 2
Unsteady Bridges Friction Slope Method= 1
Parabolic Critical Depth
Global Vel Dist= 0 , 0 , 0
Global Log Level= 0
CheckData=True
Encroach Param=-1 ,0,0, 0
Computation Interval=0.1SEC
Output Interval=1SEC
Instantaneous Interval=Max Profile
Mapping Interval=1HOUR
Computation Time Step Use Courant=        0
Computation Time Step Use Time Series=    0
Computation Time Step Count To Double=0
Computation Time Step Max Doubling=0
Computation Time Step Max Halving=0
Computation Time Step Residence Courant=0
Run HTab= 0
Run UNet= 0
Run Sediment= 0
Run PostProcess= 0
Run WQNet= 0
Run RASMapper=-1
UNET Theta= 0
UNET Theta Warmup= 0
UNET ZTol= 0
UNET ZSATol= 0
UNET MxIter= 0
UNET Max Iter WO Improvement= 0
UNET MaxInSteps= 0
UNET DtIC= 0
UNET DtMin= 0
UNET MaxCRTS= 0
UNET WFStab= 0
UNET SFStab= 0
UNET WFX= 1
UNET SFX= 1
UNET Gravity=32.174
UNET 1D Methodology=Finite Difference
UNET DSS MLevel= 1
UNET Pardiso=0
UNET DZMax Abort= 0
UNET Use Existing IB Tables= 0
UNET Froude Reduction=False
UNET Froude Limit= 0
UNET Froude Power= 0
UNET D1 Cores= 0
UNET WindReference=Eulerian
UNET WindDragFormulation=Hsu (1988)
UNET D2 Coriolis=0
UNET D2 Cores= 0
UNET D2 Theta= 1
UNET D2 Theta Warmup= 1
UNET D2 Z Tol= 0.01
UNET D2 Volume Tol= 0.01
UNET D2 Max Iterations= 20
UNET D2 Equation= 0
UNET D2 RampUpFraction=0.1
UNET D2 TimeSlices= 1
UNET D2 Turbulence Formulation=Non-Conservative (original)
UNET D2 Eddy Viscosity=0.3
UNET D2 Transverse Eddy Viscosity=0.1
UNET D2 Smagorinsky Mixing=0
UNET D2 BCVolumeCheck=0
UNET D2 Cores=0
UNET D2 SolverType=PARDISO (Direct)
UNET D2 Minimum Iterations= 2147483647
UNET D2 Maximum Iterations= 2147483647
UNET D2 Restart Number= 10
UNET D2 Relaxation Coeff=1.3
UNET D2 SOR Precondition Iterations= 10
UNET D2 ILUT Maximum Fill= 8
UNET D2 ILUT Tolerance=1E-08
UNET D1D2 MaxIter= 0
UNET D1D2 ZTol=0.01
UNET D1D2 QTol=0.1
UNET D1D2 MinQTol=1
DSS File=dss
Write IC File= 0
Write IC File at Fixed DateTime=0
Write IC File at Sim End=0
Echo Input=False
Echo Parameters=False
Echo Output=False
Write Detailed= 0
HDF Write Warmup=0
HDF Write Time Slices=0
HDF Flush=0
HDF Compression= 1
HDF Chunk Size= 1
HDF Spatial Parts= 1
HDF Use Max Rows=0
HDF Fixed Rows= 1
Calibration Method= 0
Calibration Iterations= 20
Calibration Max Change=0.05
Calibration Tolerance=0.2
Calibration Maximum=1.5
Calibration Minimum=0.5
Calibration Optimization Method= 1
WQ AD Non Conservative
WQ ULTIMATE=-1
WQ Max Comp Step=1HOUR
WQ Output Interval=15MIN
WQ Output Selected Increments= 0
WQ Output face flow=0
WQ Output face velocity=0
WQ Output face area=0
WQ Output face dispersion=0
WQ Output cell volume=0
WQ Output cell surface area=0
WQ Output cell continuity=0
WQ Output cumulative cell continuity=0
WQ Output face conc=0
WQ Output face dconc_dx=0
WQ Output face courant=0
WQ Output face peclet=0
WQ Output face adv mass=0
WQ Output face disp mass=0
WQ Output cell mass=0
WQ Output cell source sink temp=0
WQ Output nsm pathways=0
WQ Output nsm derived pathways=0
WQ Create Restart=0
WQ Fixed Restart=0
WQ System Summary=0
WQ Write To DSS=0
Sorting and Armoring Iterations= 10
XS Update Threshold= 0.02
Bed Roughness Predictor= 0
Hydraulics Update Threshold= 0.02
Energy Slope Method= 1
Volume Change Method= 1
Sediment Retention Method= 0
Sediment TS Multiplier= 1
Warm Up Method= 0
XS Weighting Method= 0
Number of US Weighted Cross Sections= 1
Number of DS Weighted Cross Sections= 1
Upstream XS Weight=0
Main XS Weight=1
Downstream XS Weight=0
Number of DS XS's Weighted with US Boundary= 1
Upstream Boundary Weight= 1
Weight of XSs Associated with US Boundary= 0
Number of US XS's Weighted with DS Boundary= 1
Downstream Boundary Weight= 0.5
Weight of XSs Associated with DS Boundary= 0.5
Percentile Method= 0
Sediment Output Level= 3
Mass or Volume Output= 0
Output Increment Type= 1
Profile and TS Output Increment= 1
Transport Output Increment 1
XS Output Flag= 0
XS Output Increment= 10
Read HDF5 Sediment Hotstart= 0
Sediment Hotstart Type= 0
Write Gradation File= 0
Read Gradation Hotstart= 0
Write HDF5 File= 1
Write Binary Output= 1
Write DSS Sediment File= 0
DSS Sediment Output Type= 1
SV Curve= 0
Specific Gage Flag= 0
Subcell Erosion Methods= 0
Subcell Deposition Methods= 0
Advection Scheme= 1
Matrix Solver= 0
Implicit Weighting Factor= 1
Maximum Outer Loop Convergence Iterations= 5
Convergence Maximum Absolute= 0.001
Convergence RMSE= 0.0001
Grain Fractions Max Abs Error= 0.001
Max Subgrid Regions= 1
Max Subgrid Length Scale= 3.402823E+38
Initial Layer Thickness= 3.402823E+38
Min Layer Thickness= 3.402823E+38
Max Layer Thickness= 3.402823E+38
Number of Layers= 5

--- MLLSTNCK.f01 (steady flow) ---

Flow Title=Flow
Program Version=6.10
Number of Profiles= 6
Profile Names=01pct,10pct,04pct,02pct,0_2pct,01plus
River Rch & RM=MLLSTNCK,Main            ,9751
     526     277     369     445     735     777
River Rch & RM=MLLSTNCK,Main            ,9377
     574     303     403     486     801     848
River Rch & RM=MLLSTNCK,Main            ,6637
     636     337     448     539     886     940
River Rch & RM=MLLSTNCK,Main            ,5514
     803     430     568     681    1110    1190
River Rch & RM=MLLSTNCK,Main            ,4994
     893     490     633     759    1240    1320
Boundary for River Rch & Prof#=MLLSTNCK,Main            , 1
Up Type= 0
Dn Type= 3
Dn Slope=0.01397
Boundary for River Rch & Prof#=MLLSTNCK,Main            , 2
Up Type= 0
Dn Type= 3
Dn Slope=0.01397
Boundary for River Rch & Prof#=MLLSTNCK,Main            , 3
Up Type= 0
Dn Type= 3
Dn Slope=0.01397
Boundary for River Rch & Prof#=MLLSTNCK,Main            , 4
Up Type= 0
Dn Type= 3
Dn Slope=0.01397
Boundary for River Rch & Prof#=MLLSTNCK,Main            , 5
Up Type= 0
Dn Type= 3
Dn Slope=0.01397
Boundary for River Rch & Prof#=MLLSTNCK,Main            , 6
Up Type= 0
Dn Type= 3
Dn Slope=0.01397
DSS Import GetInterval= 0
DSS Import GetPeak= 0
DSS Import FillOption= 0

--- MLLSTNCK.g01 (geometry) ---

Geom Title=Geometry
Program Version=6.10

River Reach=MLLSTNCK        ,Main
Reach XY= 30
2184148.37913381414824.7523151212183933.89646034414450.381896516
2183975.39341866414370.6975532332183861.59501148414089.129234795
2184113.88633478413311.8886595772183601.38520287412543.089407105
2183699.93934458412451.5285350112183652.63901596412341.957030186
  2183823.738912412339.6569058082183865.24751784412208.832397108
 2184191.5723374412070.4289132982184325.24568616412105.865883031
     2184283.213      411804.3092184889.58419224411601.916711634
     2185171.798       411681.97     2185170.001      411821.493
     2185253.822      411852.789     2185558.223      411509.778
     2185749.196      411743.8672185939.85559069  411731.0945024
     2185947.989      411919.022 2186033.9131035411989.295670425
2186305.98905637411934.360825917      2186757.31      412069.778
 2187323.7879944411570.8501746092187680.56252765411429.845086041
2187944.45216331411768.8576855382188063.50058892  411813.3277392
2188215.12923395411688.767637634     2188326.223      411827.719

Type RM Length L Ch R = 1 ,9751    ,236.4,236.4,236.4
XS GIS Cut Line= 3
2184392.69753511414764.4952761642184042.16048703414834.225764223
2183874.43039413415024.571150548
#Sta/Elev= 30
       0 2281.08    24.8 2279.13    45.4 2275.49    57.6 2274.11    86.1 2267.02
   109.9 2263.43   167.7 2260.57   171.8 2260.06   175.9 2260.27   184.7 2262.11
   208.5 2262.81   220.8 2261.94   232.3 2262.04   244.2 2260.14   253.4 2259.24
   256.62260.072   261.5 2261.77   265.6 2261.88   290.2 2260.78   334.4 2261.17
   377.3 2260.21   409.1 2260.44     427  2259.7   457.2 2260.87   511.7 2261.49
   539.5 2262.64   559.3  2264.4   573.5 2266.32   584.8 2268.66   611.1    2273
#Mann= 3 ,-1,0
       0     .05       0   244.2    .045       0   256.6     .05       0
#XS Ineff= 2 , 0
          206.27 2263.56
Permanent Ineff=
       F       F
Bank Sta=244.2,256.6
XS Rating Curve= 0 ,0
Exp/Cntr(USF)=0,0
Exp/Cntr=0.3,0.1

Type RM Length L Ch R = 1 ,9514    ,137.3,137.8,136.7
XS GIS Cut Line= 3
2184157.12156194414553.4192041992183896.88398631414678.669402499
2183789.75830037414895.630379793
#Sta/Elev= 30
       0 2267.44     8.7 2267.49    36.3 2266.64    63.2 2264.77    72.1 2263.75
    82.5 2261.82    87.4 2260.79    94.3 2258.83    98.7 2258.14   105.4 2257.71
     112 2256.71   120.9 2256.96   125.42256.745   135.4 2256.72   141.4 2257.14
   156.4 2257.13   178.6 2256.28   196.4 2257.09   209.7  2256.4   245.2 2255.76
   273.2 2256.03   288.8 2256.67   318.1 2257.18     345 2257.96   362.9 2258.97
   385.3 2259.72   429.9 2259.86   474.5 2260.77   518.2 2262.12   530.8 2262.94
#Mann= 3 ,0,0
       0     .05       0   125.4    .045       0   135.4     .05       0
Bank Sta=125.4,135.4
XS Rating Curve= 0 ,0
Exp/Cntr(USF)=0,0
Exp/Cntr=0.3,0.1

Type RM Length L Ch R = 1 ,9377    ,187.3,190.2,189.5
XS GIS Cut Line= 5
2184171.88891369 414534.927697722184038.66454407414463.810615081
2183862.72491763414554.1752102342183787.71481513414676.326601751
2183757.58471143414805.956647442
#Sta/Elev= 30
       0 2267.06    17.8 2266.55    54.1 2264.06    71.7  2262.1    92.7 2259.13
   110.5 2257.31   126.6 2256.44   153.8 2255.72   167.3 2255.02   174.7 2255.03
   183.6  2253.9   190.12253.424   194.3 2253.06   199.32253.395   216.8 2253.68
   225.2  2254.7   234.1 2254.93   241.6 2254.62   266.2  2254.6   288.7 2253.65
   302.4  2253.9   320.4 2253.41   338.1 2254.34   381.9 2254.79   419.7 2255.62
   455.6 2257.64   489.5 2258.07     530 2257.89   579.1 2259.08   625.2 2260.63
#Mann= 3 ,-1,0
       0     .05       0   190.1    .045       0   199.3     .05       0
Bank Sta=190.1,199.3
XS Rating Curve= 0 ,0
Exp/Cntr(USF)=0,0
Exp/Cntr=0.3,0.1

Type RM Length L Ch R = 1 ,9186    ,245.1,249.7,253.8
XS GIS Cut Line= 4
2184124.18558795414459.7480367052183997.02665395414350.407552062
2183839.90032787 414399.81325253 2183749.1882221414374.705437538
#Sta/Elev= 30
       0 2256.06    15.8 2254.71    28.5 2254.19    83.7 2253.88   116.1 2252.89
   172.8 2252.14   176.9 2251.69   181.2 2251.81   185.4 2251.27   188.42250.566
   193.8 2249.79   201.22250.384   206.3 2250.71   210.5 2251.19   214.7 2252.02
   218.9 2252.29   273.4  2250.3     281 2250.52   298.6 2251.55   311.2  2251.6
   332.4 2252.15   357.1 2251.88   360.3 2252.35   363.6 2253.17   370.1 2255.16
   377.8 2257.96   402.7 2268.84   412.3 2273.49   418.8 2276.07   426.5 2278.52
#Mann= 4 ,-1,0
       0     .05       0   188.4    .045       0   201.2     .05       0
  402.41      .1       0
Bank Sta=188.4,201.2
XS Rating Curve= 0 ,0
Exp/Cntr(USF)=0,0
Exp/Cntr=0.3,0.1

Type RM Length L Ch R = 1 ,8937    ,116.2,117.2,117.2
XS GIS Cut Line= 4
2184165.95730307414181.8521579072183989.73728831414138.206018902
2183824.49405798414136.6409965372183688.86057387414147.348903177
#Sta/Elev= 30
       0 2253.46    22.4 2253.09    59.5 2251.69     179 2249.37   215.1  2248.4
   243.1 2248.31   259.1 2248.75   271.1 2247.82   279.2 2247.72   296.32247.034
   307.1 2246.65   312.52247.407   315.1 2247.77   331.1 2248.03   338.7 2249.12
   343.1 2250.07   347.1 2251.25   355.3 2255.03   367.2 2261.68   375.2 2266.74
   379.2 2269.83   392.2 2278.07   399.3 2281.59   403.3 2283.95   418.3  2291.4
   433.1 2299.13   447.4 2305.44   451.4 2306.98   455.5  2308.1   482.9 2317.84
#Mann= 4 ,-1,0
       0     .05       0  271.54      .1       0   296.3    .045       0
   312.5      .1       0
Bank Sta=296.3,312.5
XS Rating Curve= 0 ,0
Exp/Cntr(USF)=0,0
Exp/Cntr=0.3,0.1

Type RM Length L Ch R = 1 ,8819    ,227.4,228.5,228.6
XS GIS Cut Line= 3
2184188.62374101 414072.901979652184016.21609446414029.218881745
2183682.20040002414012.536769791
#Sta/Elev= 30
       0 2253.57   177.9 2248.41   219.9 2246.33     239 2246.06     274 2246.48
     282 2246.32     290 2245.51     298 2246.23   306.1 2245.98   310.1 2246.32
   314.1 2246.27     317 2245.67   326.1 2244.98   334.3 2245.62     342 2246.42
   350.1 2249.83   354.1 2252.34   362.1 2259.76   370.1 2266.54   374.1 2270.54
   378.1 2273.53   387.7 2279.28   398.2 2283.67   418.2 2293.21   426.2 2296.74
   433.5 2299.13   454.2 2307.48   466.3 2310.98   498.3 2322.42   512.3 2325.73
#Mann= 6 ,-1,0
       0     .05       0  287.86      .1       0     317    .045       0
   334.3      .1       0  387.86     .05       0  487.86      .1       0
Bank Sta=317,334.3
XS Rating Curve= 0 ,0
Exp/Cntr(USF)=0,0
Exp/Cntr=0.3,0.1

Type RM Length L Ch R = 1 ,8591    ,255.4,260,259.9
XS GIS Cut Line= 3
2184257.42908315413845.6524018132184072.31421159413818.422167895
2183755.70010365413812.768344539
#Sta/Elev= 30
       0 2254.68    17.4 2254.14    57.9 2252.06    94.3 2249.23   114.5 2248.07
   166.8 2246.78   211.3 2246.25   259.2 2244.13   274.9 2243.01   283.3 2243.72
   287.3 2243.71   295.3 2243.38   303.3 2243.54   319.3 2243.22   322.1 2242.84
   327.3 2242.21   333.9 2242.92   339.3 2243.36   347.3 2243.21   359.3  2243.8
   363.3 2244.63   375.3 2251.57   383.3 2257.81   403.3  2271.3   422.2 2280.63
     440 2287.99   463.3 2295.03   475.3  2297.6   487.4 2301.75   503.8 2306.67
#Mann= 3 ,-1,0
       0     .05       0   322.1    .045       0   333.9     .05       0
Bank Sta=322.1,333.9
XS Rating Curve= 0 ,0
Exp/Cntr(USF)=0,0
Exp/Cntr=0.3,0.1

Type RM Length L Ch R = 1 ,8331    ,252.3,250.4,244.6
XS GIS Cut Line= 3
2184222.19529648413668.0311416882183855.13301958413548.930474674
2183725.54637908413607.346095931
#Sta/Elev= 30
       0 2250.16    27.4 2248.73    56.8 2245.56    69.4 2244.65   107.3 2243.29
   170.3 2240.46   177.7 2240.51   180.72240.141   187.2 2239.38   199.62240.089
   208.2 2240.08   216.6 2240.91   220.8 2240.93   254.7 2239.82   304.9 2239.07
   317.5 2239.73   384.7 2240.84   412.5 2243.28   424.2 2244.87   430.7 2244.98
   435.2 2245.42   450.6 2249.88   468.1 2257.22     473 2259.43   485.1  2265.9
   494.4 2268.88   503.2 2274.16   512.3 2277.02   521.4 2279.16     528 2280.33
#Mann= 3 ,-1,0
       0     .05       0   180.7    .045       0   199.6     .05       0
Bank Sta=180.7,199.6
XS Rating Curve= 0 ,0
Exp/Cntr(USF)=0,0
Exp/Cntr=0.3,0.1

Type RM Length L Ch R = 1 ,8081    ,258.8,255.9,249
XS GIS Cut Line= 4
2184313.02937974413440.9302790262184177.79079886413377.100205037
2183922.64298923413376.3032546992183717.38602737413552.070549585
#Sta/Elev= 30
       0 2250.23    15.5 2250.24    27.5 2249.75    80.6 2244.95   111.9 2241.42
   167.3 2237.41   179.2 2236.98   195.2 2237.27   211.2 2236.53   219.2 2237.07
   222.52236.615   227.2 2236.28   231.92236.579   239.2    2237   367.2 2237.08
   418.5 2236.44   432.6 2235.75   492.2 2237.91   526.2 2239.64   555.4  2240.5
     587  2242.7   597.1 2244.63   602.8 2244.84   605.6 2245.38   619.8 2249.72
     634 2257.03   639.7 2259.24     652 2265.07   664.3 2268.96   674.9 2271.13
#Mann= 3 ,-1,0
       0     .05       0   222.5    .045       0   231.9     .05       0
#XS Ineff= 2 , 0
          184.21 2241.25
Permanent Ineff=
       F       F
Bank Sta=222.5,231.9
XS Rating Curve= 0 ,0
Exp/Cntr(USF)=0,0
Exp/Cntr=0.3,0.1

Type RM Length L Ch R = 1 ,7825    ,221.6,229.7,233.6
XS GIS Cut Line= 4
2184228.03398398 413140.828336132184072.83800047413129.703463349
2183826.25218368 413256.657953092183721.71331596413416.361076225
#Sta/Elev= 30
       0  2240.8   100.1 2237.88   178.8 2236.33   183.3 2236.04   194.3 2234.53
   205.8 2233.79   215.1 2233.74   218.1 2233.31  219.832232.664     221 2232.23
   223.8 2231.59     2282232.665   232.9 2233.28   237.3 2233.45   259.8 2233.59
   277.5 2233.32   291.3 2233.32   336.3 2234.09   345.3 2234.08   372.3 2234.81
   427.3 2234.94   457.5 2236.05   482.9 2237.43   509.9 2238.31   517.1 2238.15
   524.4 2238.28   553.3 2239.78   581.8 2240.52   611.1 2241.88   623.8 2242.79
#Mann= 3 ,0,0
       0     .05       0  219.83    .045       0     228     .05       0
#XS Ineff= 2 , 0
                          371.89         2235.75
Permanent Ineff=
       F       F
Bank Sta=219.83,228
XS Rating Curve= 0 ,0
Exp/Cntr(USF)=0,0
Exp/Cntr=0.3,0.1

Type RM Length L Ch R = 1 ,7595    ,172.6,166.2,159.7
XS GIS Cut Line= 6
 2184211.1766586412955.2968243112184026.68931651412936.881196959
2183905.96184091413000.8159864522183887.55445063 412998.33806853
2183672.29232096413111.0253701912183593.23229392413214.938256398
#Sta/Elev= 30
       0 2236.53    35.2 2234.99    55.3 2233.74   119.6 2231.83   135.7 2231.82
   172.8 2231.13   192.8 2231.39   234.8 2230.83   247.1 2230.99   255.5 2230.69
   274.2 2230.96   279.2 2230.66   296.9  2230.5   317.7 2230.57   320.6 2230.41
   326.8 2229.46   331.9 2228.84   336.92229.459   344.4  2230.4   365.9 2230.67
   383.7 2230.46   394.1 2229.67   407.6 2229.25   415.7 2229.34   479.9 2231.97
   540.8 2232.31     597 2233.82   656.6 2234.16     663 2234.49   714.1 2235.41
#Mann= 3 ,0,0
       0     .05       0   326.8    .045       0   336.9     .05       0
Bank Sta=326.8,336.9
XS Rating Curve= 0 ,0
Exp/Cntr(USF)=0,0
Exp/Cntr=0.3,0.1

Type RM Length L Ch R = 1 ,7429    ,176.1,178.8,177.1
XS GIS Cut Line= 5
2184178.62210411412851.8042161662184034.04172215412731.723177346
2183956.76632783412779.3959360672183687.18980428412950.072445221
2183584.50866068413124.744898634
#Sta/Elev= 30
       0 2233.26    29.2 2232.12    54.7 2230.57   107.2 2229.38   122.8 2229.13
   139.9  2229.2   159.2  2228.8   187.9 2227.67     223 2227.54   312.6 2227.84
     379 2227.56     412 2228.12   413.8    2228   417.82227.161   422.5 2226.22
   429.7 2227.08   439.9 2228.21   442.7 2228.29   471.8 2227.69   487.8    2227
   506.6 2227.72   516.2 2227.14   528.8 2227.77     554 2229.71     573  2230.8
   629.2 2231.29   674.8  2232.2   701.6 2233.14   789.3 2233.38   800.4 2233.82
#Mann= 3 ,0,0
       0     .05       0   417.8    .045       0   429.7     .05       0
#XS Ineff= 2 , 0
          403.94 2229.69
Permanent Ineff=
       F       F
Bank Sta=417.8,429.7
XS Rating Curve= 0 ,0
Exp/Cntr(USF)=0,0
Exp/Cntr=0.3,0.1

Type RM Length L Ch R = 1 ,7250    ,61,60.2,59.5
XS GIS Cut Line= 4
2184153.60512692412755.993070889 2183930.0443282412631.135319912
2183591.52509846412833.6796790862183545.12517221412976.656196013
#Sta/Elev= 30
       0 2229.84    38.3 2228.81    94.3 2228.03   125.3 2227.27     137 2226.76
   175.7 2225.92   194.4 2225.59   226.1 2225.47   258.2 2224.82   281.5 2224.78
   305.6 2225.29   330.2 2225.46   413.5 2225.48   448.5 2226.05   457.2 2226.45
   478.2 2226.42   506.8 2225.46   514.6 2225.17  517.682225.454   523.9 2225.79
   540.5 2225.41   559.3 2224.15   565.1 2223.97   626.5 2225.92   650.6 2227.54
   662.3 2229.02   671.1 2229.78   696.3 2230.99     713 2231.41   800.9 2232.38
#Mann= 3 ,0,0
       0     .05       0   506.8    .045       0  517.68     .05       0
#XS Ineff= 2 , 0
           469.3 2227.95
Permanent Ineff=
       F       F
Bank Sta=506.8,517.68
XS Rating Curve= 0 ,0
Exp/Cntr(USF)=0,0
Exp/Cntr=0.3,0.1

Type RM Length L Ch R = 1 ,7190    ,136.5,136,133.6
XS GIS Cut Line= 6
2184151.52813507412745.5285691462183932.85221257412625.753356419
2183851.67132421 412587.488565662183829.76535965412604.065599322
2183523.35302094412822.0680262622183515.82473025413022.425366525
#Sta/Elev= 30
       0 2229.59    44.9 2228.57    94.1 2227.92   140.6 2226.42   186.3 2225.53
   226.7 2225.39   272.2  2224.2   320.8 2223.64   377.1 2223.82   445.9 2224.85
   503.3 2225.25   527.2  2225.1   540.6 2225.34   547.9 2225.18   552.82224.711
     555 2224.44  558.772224.698   564.9 2225.31   583.6 2225.07   603.7 2223.52
   623.8    2223     663  2223.8   687.6 2223.98   724.2 2225.17   742.6 2226.45
   773.7 2230.25   789.7 2231.44     849 2231.78   925.5 2232.81   943.1  2232.7
#Mann= 3 ,0,0
       0     .05       0   552.8    .045       0  558.77     .05       0
#XS Ineff= 2 , 0
          539.18 2226.16
Permanent Ineff=
       F       F
Bank Sta=552.8,558.77
XS Rating Curve= 0 ,0
Exp/Cntr(USF)=0,0
Exp/Cntr=0.3,0.1

Type RM Length L Ch R = 1 ,7054    ,151.9,170.9,188.2
XS GIS Cut Line= 6
 2184141.1158057412731.9828251522183796.13262639412554.596331113
2183649.85895709412574.3792454042183588.11228521412618.740931998
2183435.84379339 412776.404764082183413.66295009412836.952471457
#Sta/Elev= 30
       0 2229.16    32.7  2228.5    50.1 2228.51    91.6 2227.66   100.6 2227.12
   136.8 2226.07   168.5 2225.56   222.8 2225.19   245.2 2224.42   267.5 2224.05
   309.8 2223.59   420.2 2223.38   445.6 2223.74   521.1 2223.93   547.4 2223.66
  555.012222.518   557.3 2222.13   567.2 2221.82     576  2222.5     582 2223.36
   584.6 2223.45     615 2223.56   647.2 2222.46   664.2 2222.99   712.3 2222.62
   770.7 2222.77   844.4 2224.98   852.8 2225.49   876.3 2228.34   895.3 2229.89
#Mann= 3 ,0,0
       0     .05       0  555.01    .045       0     576     .05       0
#XS Ineff= 2 ,-1
       0  514.37  2224.9  615.21  786.562225.196
Permanent Ineff=
       F       F
Bank Sta=555.01,576
XS Rating Curve= 0 ,0
Exp/Cntr(USF)=0,0
Exp/Cntr=0.3,0.1

Type RM Length L Ch R = 1 ,6883    ,228.9,246.2,254.6
XS GIS Cut Line= 5
2184152.63006667412726.5958461062183906.47499352412601.774066368
2183666.42337509412464.2863337862183587.06594926412459.094726488
2183257.02805676412261.071990988
#Sta/Elev= 30
       0 2229.28    90.7 2227.81   135.8 2226.15   229.2 2225.27   301.7 2223.65
   500.9 2222.66   504.5 2222.53   512.6 2220.55   527.6 2219.78  534.122220.483
   541.4 2221.36   578.9  2220.7     603  2221.9     619 2220.61     627 2221.29
   650.2 2220.49   654.2 2220.02   659.2 2218.24   667.7 2217.94   705.5 2219.41
   756.8 2218.66   780.1 2219.11   798.3  2218.3   813.5 2220.13   840.8 2219.31
   882.8 2220.31   912.6 2224.33   971.4 2223.61   994.3 2227.23    1017 2234.39
#Mann= 3 ,0,0
       0     .05       0   512.6    .045       0  534.12     .05       0
#XS Ineff= 1 ,-1
  627.56  814.132224.726
Permanent Ineff=
       F
Bank Sta=512.6,534.12
XS Rating Curve= 0 ,0
Exp/Cntr(USF)=0,0
Exp/Cntr=0.3,0.1

Type RM Length L Ch R = 1 ,6637    ,117.4,110.8,92.3
XS GIS Cut Line= 4
2184022.41930408412657.117461989  2183722.047739412448.711511893
2183717.59778989412310.0214312242183630.82378219412184.681197892
#Sta/Elev= 30
       0 2225.92    24.6 2225.53    75.8 2225.38     105 2224.44   148.8 2223.56
   238.5 2223.17   247.7 2222.96   280.2  2223.1   337.9 2222.75     363 2222.91
   393.1 2219.98   448.4 2218.81   457.2 2217.61   461.2 2216.85   465.2 2216.58
   471.6 2217.56   481.2 2218.04   489.2 2219.05   497.2 2219.59   517.5 2219.14
   549.2 2219.47   554.9 2219.86   558.9 2220.48   563.8 2221.64   569.2 2223.31
   589.3 2230.23     598 2232.98   631.9 2245.19   647.4 2252.23   656.8 2255.97
#Mann= 4 ,-1,0
       0     .05       0   457.2    .045       0   471.6     .05       0
  624.35      .1       0
Bank Sta=457.2,471.6
XS Rating Curve= 0 ,0
Exp/Cntr(USF)=0,0
Exp/Cntr=0.3,0.1

Type RM Length L Ch R = 1 ,6526    ,225.1,232.1,232.7
XS GIS Cut Line= 4
2184159.48847474412717.3470064552183974.21648791412542.425323493
2183861.92476886412393.4576064392183701.57026592412179.191188893
#Sta/Elev= 30
       0 2229.31    81.8    2228   157.6 2225.23     209  2225.1   285.7 2223.38
     360 2222.91     411 2222.16     431 2222.53   436.7    2222   444.3 2221.98
   459.9 2220.66   466.7 2219.82   477.7 2217.76   491.7 2217.32   499.12216.404
   506.6  2215.3   511.4 2215.06   524.4 2216.35   528.5 2216.92   536.6 2218.53
     540 2218.65   551.1  2218.5   565.7 2219.09   581.6  2219.2     600 2218.62
     620 2218.64   631.6 2219.13   646.5 2220.84   657.9 2223.98     709 2242.02
#Mann= 4 ,-1,0
       0     .05       0   499.1    .045       0   524.4     .05       0
   528.5      .1       0
Bank Sta=499.1,524.4
XS Rating Curve= 0 ,0
Exp/Cntr(USF)=0,0
Exp/Cntr=0.3,0.1

Type RM Length L Ch R = 1 ,6294    ,166.4,166.4,165.6
XS GIS Cut Line= 5
2184164.32552037 412660.991502192184021.31175886412448.847411475
2183985.13882496412275.8955712612183919.57538227412141.377473317
2183718.83965192412046.434115533
#Sta/Elev= 30
       0 2228.46   100.8 2227.14   143.4 2225.17     193    2224   276.8 2223.49
   333.2  2222.3   390.4 2222.38     412 2221.54   447.3 2222.01   453.4 2221.64
   471.2 2218.66   502.3 2217.96   515.7 2218.29   520.1 2217.89   523.2 2216.95
   524.52216.532     529 2215.06   533.5 2214.55   542.4 2215.03     546 2216.62
     549 2217.85   553.4  2218.7   581.9 2219.69   608.9 2221.66   630.9 2225.44
     645  2229.2   692.1 2244.13   747.1 2256.86   767.4 2260.76   804.2 2270.31
#Mann= 5 ,-1,0
       0     .05       0   523.2      .1       0   524.5    .045       0
     546      .1       0   630.9     .05       0
Bank Sta=524.5,546
XS Rating Curve= 0 ,0
Exp/Cntr=0.3,0.1

Type RM Length L Ch R = 1 ,6127    ,253.8,253.9,249
XS GIS Cut Line= 4
2184336.10875452412362.6940948342184132.34266681412200.374686101
 2184047.3110551 412031.728267432183870.96800234 411746.86641296
#Sta/Elev= 30
       0 2223.64    40.9 2223.31   103.5 2220.06   137.2 2219.09   211.7 2220.04
   234.4 2219.88   252.8 2220.37   264.1 2219.92   277.5 2220.44   310.7 2218.23
   328.5 2218.15   346.4 2217.41   349.4 2217.15   354.5  2215.9   358.3 2215.07
   362.6  2214.7   367.3 2214.86   371.32216.046   376.2 2217.19   389.5  2218.3
     400 2218.24   420.8 2219.03   447.7 2218.87   488.4 2217.91   523.7 2218.06
   588.8 2217.45   621.7 2217.75   678.2 2219.79   706.3 2221.97   784.4 2225.76
#Mann= 3 ,-1,0
       0     .05       0   354.5    .045       0   371.3     .05       0
#XS Ineff= 2 , 0
          298.03 2222.64     640         2222.82
Permanent Ineff=
       F       F
Bank Sta=354.5,371.3
XS Rating Curve= 0 ,0
Exp/Cntr(USF)=0,0
Exp/Cntr=0.3,0.1

Type RM Length L Ch R = 1 ,5874    ,353.9,360.1,363.6
XS GIS Cut Line= 5
2184346.30024891412360.7692564762184354.78099326412203.549703459
2184345.73775979412152.6815151612184271.13108362412018.163417217
2183993.90658871411626.827041189
#Sta/Elev= 30
       0 2223.58    35.6 2224.25   119.8  2224.1   188.3 2222.28   200.5 2222.35
   212.8 2221.86   215.8 2221.38   228.8 2217.92     236 2217.01   242.3 2216.68
   248.1  2215.7   258.9 2214.62   270.1 2215.65   281.7 2216.47   286.4 2217.54
   294.8 2217.91   368.6 2217.11   388.3 2217.71   431.8 2217.51   523.6  2215.4
     541 2215.64   579.8 2217.32   640.4 2217.34   665.6  2218.2   692.9 2220.61
   707.1 2221.28   751.4 2221.39   793.3 2222.84   819.1 2224.24   842.5 2226.59
#Mann= 3 ,-1,0
       0     .05       0   248.1    .045       0   270.1     .05       0
#XS Ineff= 2 , 0
                          648.42         2223.02
Permanent Ineff=
       F       F
Bank Sta=248.1,270.1
XS Rating Curve= 0 ,0
Exp/Cntr(USF)=0,0
Exp/Cntr=0.3,0.1

Type RM Length L Ch R = 1 ,5514    ,314.4,317.8,319.6
XS GIS Cut Line= 3
 2184654.6813565412118.3223553962184389.73353738411970.120872172
2184138.69787835411515.152860058
#Sta/Elev= 30
       0 2222.79    26.9 2221.99    76.2 2221.66   120.2 2219.25   140.4 2218.62
   202.5 2218.71   340.7 2221.12   354.9 2219.64   364.3 2219.46   370.2 2218.53
   414.4 2218.41   437.1 2216.99   458.5 2216.41   473.7 2217.03   478.3 2216.74
   485.92215.001   496.8 2212.84   510.2 2213.16     514 2214.94   520.3 2218.53
   523.9  2219.4   532.1  2219.7   633.6 2218.51   667.5 2218.64   720.8 2217.68
     750 2218.16   766.1 2219.18   776.5 2220.71   814.7 2229.78   823.2 2231.01
#Mann= 4 ,-1,0
       0     .05       0   485.9    .045       0     514     .05       0
   814.7     .06       0
#XS Ineff= 2 , 0
          334.65 2223.19
Permanent Ineff=
       F       F
Bank Sta=485.9,514
XS Rating Curve= 0 ,0
Exp/Cntr(USF)=0,0
Exp/Cntr=0.3,0.1

Type RM Length L Ch R = 1 ,5196    ,202,201.3,201.4
XS GIS Cut Line= 4
2184749.29205362412019.2938214012184618.16516822 411795.47379289
2184551.47132134411601.0442731742184542.42808788411378.354648845
#Sta/Elev= 30
       0 2224.61    72.5 2222.61   133.9 2222.47   206.4 2220.42   266.1 2220.43
   287.2 2219.15   295.7 2219.23   304.1    2218   347.8 2217.67   359.1 2215.98
   367.5 2216.16   371.8 2215.82   379.3 2213.57   384.5 2211.98   388.6 2211.63
   397.1 2212.19   400.62213.659   405.6  2217.4   409.8 2218.79   418.3 2218.85
   422.5 2219.78   439.4 2221.61   461.1  2222.6   520.9 2222.58   568.9 2223.53
   625.7  2226.3     653 2226.98     661 2228.09     673 2230.89   687.8 2235.64
#Mann= 5 ,-1,0
       0     .05       0   339.4     .06       0   379.3    .045       0
   400.6     .06       0   439.4     .05       0
#XS Ineff= 2 , 0
          297.35 2222.96
Permanent Ineff=
       F       F
Bank Sta=379.3,400.6
XS Rating Curve= 0 ,0
Exp/Cntr(USF)=0,0
Exp/Cntr=0.3,0.1

Type RM Length L Ch R = 1 ,4994    ,120,118,114.6
BEGIN DESCRIPTION:
xs 4
END DESCRIPTION:
XS GIS Cut Line= 3
2184879.28853483411903.9925945932184725.55356575411519.655171895
2184691.64144021411355.746565157
#Sta/Elev= 30
       0 2226.87      73 2225.38   148.4 2224.82   214.1 2223.59   231.4  2222.4
   248.6 2220.42   261.5 2216.12   272.3 2213.84   272.3 2213.83   278.8 2211.92
   283.1 2212.17   289.82213.789     300 2215.85   317.5 2216.19   326.1 2217.44
   334.8 2217.78   339.1 2218.58   343.4 2220.17   347.7 2221.09   361.5 2221.18
   373.5 2222.55   407.7 2224.51   481.8 2229.71   506.3 2232.69   518.6 2233.19
   534.9 2231.81   547.2 2232.19   555.4 2233.58   563.5 2235.57   581.3 2236.77
#Mann= 7 ,-1,0
       0     .05       0   272.3    .045       0   289.8     .05       0
     300     .06       0     410     .05       0  513.94      .1       0
  573.94     .05       0
Bank Sta=272.3,289.8
XS Rating Curve= 0 ,0
Exp/Cntr(USF)=0,0
Exp/Cntr=0.5,0.3

Type RM Length L Ch R = 1 ,4876    ,45.1,44.7,48.3
BEGIN DESCRIPTION:
xs 3
END DESCRIPTION:
XS GIS Cut Line= 6
2185006.59913473411865.926333957 2184983.1256136411778.965583495
2184924.36087383411689.7982840652184877.06849309411587.617771663
2184748.76162702411468.2108038152184723.54524871411348.062177782
#Sta/Elev= 30
       0 2232.79    25.6  2232.3    74.4 2229.76   151.2 2224.12     188 2223.58
   209.3 2222.44   222.5 2219.75   262.9 2215.64   271.9  2215.3   282.5 2213.48
   288.4 2212.13   294.4 2211.77   302.9 2212.21   309.2 2213.46   317.7  2215.4
     344 2215.94   369.8 2219.35   375.3 2219.18   394.9 2220.56   413.1 2224.84
   419.4  2225.6   449.9 2226.54     482 2228.98   514.6 2229.12   526.3 2229.78
   536.7 2231.84   547.3 2234.74   567.7 2238.16   596.3 2239.52   609.7 2240.75
#Mann= 8 ,-1,0
       0     .05       0      50     .06       0      70     .05       0
  273.71     .06       0   282.5    .045       0   309.2     .06       0
  405.26     .05       0  526.97      .1       0
#XS Ineff= 2 , 0
             268 2214.36     325         2214.03
Permanent Ineff=
       F       F
Bank Sta=282.5,309.2
XS Rating Curve= 0 ,0
Exp/Cntr(USF)=0,0
Exp/Cntr=0.5,0.3

Type RM Length L Ch R = 1 ,4832    ,175.9,190.2,203.2
BEGIN DESCRIPTION:
xs 2
END DESCRIPTION:
XS GIS Cut Line= 6
2185031.33339565411856.0980347762185006.11701735411762.649103416
2184917.85969329411583.9094807362184837.01895108411522.351851349
2184771.01137258 411449.669349182184756.17820887411361.412025119
#Sta/Elev= 30
       0 2232.82    19.6 2232.49    48.6 2230.89    56.9 2229.41    73.4 2224.72
    77.6 2224.31   108.5 2223.27   118.4 2224.47   123.4 2224.48   142.2 2223.31
   174.1 2222.52   187.4 2221.33   209.4 2218.12   234.5 2216.01   254.1 2213.39
   270.1 2212.29     282 2213.41   300.5 2214.03   322.3 2217.91   332.2 2218.88
   358.9 2223.19   407.8 2225.54     424 2227.48   443.7 2227.31   456.4 2229.13
     499 2231.69   507.6 2233.98   536.6 2237.43   568.4 2240.28   588.5 2241.05
#Mann= 7 ,-1,0
       0     .05       0      40     .06       0  126.79     .05       0
   254.1    .045       0     282     .06       0  389.34     .05       0
  518.98      .1       0
#XS Ineff= 2 , 0
             249    2214     287            2214
Permanent Ineff=
       F       F
Bank Sta=254.1,282
XS Rating Curve= 0 ,0
Exp/Cntr(USF)=0,0
Exp/Cntr=0.5,0.3

Type RM Length L Ch R = 1 ,4641    ,254.4,266.7,272.5
BEGIN DESCRIPTION:
xs 1
END DESCRIPTION:
XS GIS Cut Line= 4
2185027.37148298411888.1669360112185087.28290476411723.127925088
2185126.84705121411612.348315017 2185040.9363332411467.656579414
#Sta/Elev= 30
       0 2233.44    54.2 2232.71    59.2 2232.03    71.6 2227.08    96.6 2227.76
   118.1 2223.65   126.6 2222.76   169.1 2223.38   190.3 2222.57     206 2219.88
   225.8 2213.66     231 2211.93   237.7 2211.25   249.9 2211.57   255.72213.633
   262.3 2215.07   271.1    2216   283.8 2220.13   293.2 2221.79   315.5 2223.39
   352.9 2223.44     369 2224.01   399.6  2228.4     416 2231.97   431.8 2231.61
   439.5 2233.82   445.8 2237.54   450.4 2241.48   454.9 2244.23   461.5 2246.47
#Mann= 5 ,-1,0
       0     .05       0      70     .06       0  185.58     .05       0
   225.8    .045       0   255.7     .05       0
Bank Sta=225.8,255.7
XS Rating Curve= 0 ,0
Exp/Cntr(USF)=0,0
Exp/Cntr=0.3,0.1

Type RM Length L Ch R = 1 ,4375    ,308.3,291.5,274.1
XS GIS Cut Line= 5
 2185069.1964378412084.8572640972185228.58342781411792.082580337
2185254.58272405411729.9103501942185256.84353242411649.651653102
2185060.15320432411365.920202817
#Sta/Elev= 30
       0 2233.37    54.3 2232.48    98.3 2230.32   127.2 2230.73   149.9 2225.89
   154.5 2225.82   168.1 2229.84   181.8 2228.29   213.7 2226.47   222.8  2227.9
   227.4 2227.76   236.5 2226.19   250.1 2221.51   259.2 2216.11   265.6 2214.37
   273.3 2212.19   276.2 2212.22     282 2214.36   305.7 2220.91   327.5 2223.23
   588.2 2223.88   622.7 2222.53   705.5 2221.38     735 2222.73     752 2225.57
   770.1  2232.1   791.1 2236.18   800.9 2241.43   812.4 2254.22   826.3    2262
#Mann= 6 ,-1,0
       0     .05       0     190     .06       0   265.6    .045       0
     282     .06       0     300     .05       0  751.03      .1       0
Bank Sta=265.6,282
XS Rating Curve= 0 ,0
Exp/Cntr(USF)=0,0
Exp/Cntr=0.3,0.1

Type RM Length L Ch R = 1 ,4083    ,299,326,359.2
XS GIS Cut Line= 3
2185437.56977531412112.9093363562185435.75555583411707.887359836
2185076.12184567411350.854292087
#Sta/Elev= 30
       0 2231.21    91.7 2227.64   127.7 2228.16   179.7 2226.42   215.7 2226.32
   279.7 2223.18   351.6 2222.98   415.1 2221.81     427 2219.62   438.3 2213.61
   446.2 2210.83   451.9 2210.37   463.2 2211.06   470.32213.625   477.7 2217.27
   483.3 2218.96   497.2 2221.29   511.3 2222.28   601.9 2222.19   675.3  2220.7
   749.5 2222.77   808.3 2222.09   844.1 2223.36   859.2 2226.74   877.9 2234.65
   889.2 2236.05   894.8 2238.07   904.5 2245.39   907.3 2248.56   911.8 2255.62
#Mann= 5 ,-1,0
       0     .06       0     200     .05       0   438.3    .045       0
   470.3     .05       0  805.03      .1       0
Bank Sta=438.3,470.3
XS Rating Curve= 0 ,0
Exp/Cntr(USF)=0,0
Exp/Cntr=0.3,0.1

Type RM Length L Ch R = 1 ,3757    ,196.8,187.4,180.2
XS GIS Cut Line= 4
2185454.81891529412118.9916371712185445.91523788411702.486539844
2185681.94899004411530.9240297292185698.42479962411425.374217129
#Sta/Elev= 30
       0  2231.3    89.8 2227.68   125.9 2228.09   177.9 2226.32   233.9 2225.68
   273.9 2223.18   353.9 2222.62   389.9 2221.53     485 2222.31   518.3 2221.74
   536.6 2222.28   568.1 2222.14   577.6 2220.95   596.7 2214.39   617.2 2213.57
     6232212.179   628.2 2210.51   636.8 2210.22   641.9 2210.76   646.82212.249
   651.1 2214.01   659.7 2218.72   671.6 2226.83   691.2 2234.86   710.2 2241.09
   722.3 2246.83   738.5 2253.31   750.6 2256.33   770.9 2259.86   815.2 2266.04
#Mann= 7 ,-1,0
       0     .06       0     200     .05       0   586.6      .1       0
     623    .045       0   646.8      .1       0   706.6     .05       0
   718.4      .1       0
Bank Sta=623,646.8
XS Rating Curve= 0 ,0
Exp/Cntr(USF)=0,0
Exp/Cntr=0.3,0.1

Type RM Length L Ch R = 1 ,3570    ,238.2,240,242.6
XS GIS Cut Line= 3
2185485.42851062 412124.395432832185770.66657304411653.465477431
2185740.03698244411410.343102083
#Sta/Elev= 30
       0 2231.55     130 2228.02   190.7 2222.97   219.9 2221.42   242.3 2221.09
   298.5 2221.91   410.6 2220.34     420 2219.05   445.4 2211.89   449.9 2210.96
   462.1 2210.39   468.6 2210.49   475.8 2211.82   493.6 2214.51   513.5 2220.63
   518.2 2221.32   550.9 2221.98     563 2221.09   579.1 2218.74   591.2 2218.61
   639.6 2224.86   651.7 2227.77   663.8 2232.15   675.8 2237.29   716.2 2256.94
   728.5 2259.54   760.2 2263.83   772.6 2264.71   784.7 2268.55   795.6  2273.2
#Mann= 6 ,-1,0
       0     .06       0      10     .07       0     130     .05       0
   445.4    .045       0   475.8     .05       0  680.58      .1       0
Bank Sta=445.4,475.8
XS Rating Curve= 0 ,0
Exp/Cntr(USF)=0,0
Exp/Cntr=0.3,0.1

Type RM Length L Ch R = 1 ,3330    ,263.9,254.3,256.5
XS GIS Cut Line= 3
2185636.24180908412159.4628980942186013.04320388411645.896552587
 2186066.0745113411419.815715706
#Sta/Elev= 30
       0 2232.85    13.4 2232.31    32.6 2230.09    98.9 2228.44   164.7 2222.94
   204.8 2220.85   256.3    2220   315.4 2221.04   362.1 2220.52   399.7 2221.69
   459.7 2221.34   473.8 2220.49   484.1 2218.97   500.3 2215.12   508.9 2211.15
   513.8 2209.69   518.8 2209.35   533.8  2210.1   540.8 2211.26   573.4 2219.88
   578.3 2220.52   641.8 2219.67   674.7 2220.17   711.7 2222.53   752.7 2223.68
   781.5 2226.42   818.5  2234.3   830.8 2237.97   855.5 2248.92   869.2 2256.45
#Mann= 6 ,-1,0
       0     .07       0      50     .06       0     180     .05       0
   508.9    .045       0   540.8     .05       0  766.97      .1       0
Bank Sta=508.9,540.8
XS Rating Curve= 0 ,0
Exp/Cntr(USF)=0,0
Exp/Cntr=0.3,0.1

Type RM Length L Ch R = 1 ,3076    ,390,375.4,373.3
XS GIS Cut Line= 4
2185874.10117844412183.9549887552185954.42965358412022.697947388
2186131.66586521411771.497017521 2186222.3773121411450.518051579
#Sta/Elev= 30
       0 2233.54    34.4 2233.12    61.2 2228.68    83.5 2228.35    96.9 2226.99
   114.8 2226.43   132.7 2224.42   179.7 2223.46   195.8 2219.63   206.5 2217.64
   225.6 2211.21   235.9 2209.43   252.6 2208.46     260  2209.2   264.82211.079
   273.4 2213.81   294.6 2217.15   305.9 2220.45   311.7 2221.36   348.5 2220.96
   486.7  2223.7     545 2223.51   577.3 2222.25   618.9 2222.36   656.3 2223.26
   685.4 2224.78     707  2227.2   743.6 2232.55     781 2241.22   821.1 2254.32
#Mann= 6 ,-1,0
       0     .05       0      80     .06       0  190.16     .05       0
   225.6    .045       0   264.8     .05       0  747.59      .1       0
Bank Sta=225.6,264.8
XS Rating Curve= 0 ,0
Exp/Cntr(USF)=0,0
Exp/Cntr=0.3,0.1

Type RM Length L Ch R = 1 ,2700    ,316.6,311.1,297.5
XS GIS Cut Line= 3
2186267.03525519412131.5516836642186412.17357023411802.199353394
2186494.51165279411504.944919717
#Sta/Elev= 30
       0  2230.7    37.6 2230.11    93.7 2226.01   116.2 2225.14   120.6 2224.36
     125  2221.6   129.4 2219.76   142.5 2219.22   151.2  2214.8   155.6 2213.36
   168.7 2211.59   181.8  2211.8   184.7 2210.74   190.8 2208.41   199.9 2208.72
   212.4 2210.71   221.1 2216.33   230.2 2220.11   234.3 2221.44     243 2222.42
   373.4 2224.53   461.5 2224.41     581 2227.88   593.4 2229.84   605.9 2233.35
   614.2 2234.62   630.8 2238.24   647.4 2242.39     663 2247.04   668.4  2247.8
#Mann= 6 ,-1,0
       0     .05       0     130     .06       0   184.7    .045       0
   212.4     .06       0     230     .05       0  649.91      .1       0
Bank Sta=184.7,212.4
XS Rating Curve= 0 ,0
Exp/Cntr(USF)=0,0
Exp/Cntr=0.3,0.1

Type RM Length L Ch R = 1 ,2389    ,304.1,294.2,281.2
XS GIS Cut Line= 3
2186617.32099628412233.4276163332186604.76094979411810.572717722
2186582.43197825411504.944919717
#Sta/Elev= 30
       0 2230.46    44.3 2230.66   100.3  2227.9   104.3 2226.84   112.3 2221.32
   116.3 2219.36   132.3 2218.17   140.3 2211.85   144.3 2209.45   148.3 2207.61
   156.3 2206.57   164.6 2207.06   172.3 2209.52   172.3 2209.53   180.3 2214.32
   188.3 2217.59   208.3 2219.18   260.4 2220.12   288.9 2221.57   344.4  2223.1
   372.4 2222.95   400.4 2224.09   468.6  2225.4   500.6 2225.02   545.1 2226.97
   588.9 2227.68   612.9 2228.98     637 2231.37   657.1 2234.97   729.5 2257.02
#Mann= 6 ,-1,0
       0     .05       0     120     .06       0   144.3    .045       0
   172.3     .06       0     220     .05       0  713.04      .1       0
Bank Sta=144.3,172.3
XS Rating Curve= 0 ,0
Exp/Cntr(USF)=0,0
Exp/Cntr=0.3,0.1

Type RM Length L Ch R = 1 ,2095    ,317.7,317.8,312.4
XS GIS Cut Line= 3
2187006.68243758412184.5829910812186818.28174018411909.657528948
2186724.77917184411524.482769818
#Sta/Elev= 30
       0 2232.73    84.8 2228.99   133.7 2225.23   138.9  2223.8   145.2 2220.15
   148.1 2219.36   159.3 2218.77   164.1 2217.63   173.8 2212.16   183.5  2208.5
   188.4 2205.81     197  2205.1   199.9 2205.29   214.3 2208.39   223.8 2215.03
   236.9 2220.31   243.1 2220.97   314.5 2221.03   345.4  2222.3   362.6 2223.49
   399.6 2223.99   436.7 2225.32   562.6 2226.19   581.1 2226.71   601.3 2227.95
   630.5  2231.4   650.1 2235.62   683.7 2244.64   712.5  2253.3   729.6 2259.08
#Mann= 5 ,-1,0
       0     .05       0      90     .06       0   183.5    .045       0
   214.3     .05       0  729.65      .1       0
Bank Sta=183.5,214.3
XS Rating Curve= 0 ,0
Exp/Cntr(USF)=0,0
Exp/Cntr=0.3,0.1

Type RM Length L Ch R = 1 ,1777    ,278.7,282.5,283.2
XS GIS Cut Line= 3
2187231.36771374411962.6888363642187006.68243758411703.114542168
2186842.00627244411474.242583844
#Sta/Elev= 30
       0 2227.66    44.3 2226.13   102.5 2222.44   142.3 2221.63   145.1 2221.32
   153.6 2218.26   171.3  2217.5   194.3 2207.67   201.8 2205.04   208.3  2204.4
   224.2 2206.45   227.4 2207.66   230.2 2209.12   240.1  2216.1   245.4 2218.79
     250 2219.92   255.7 2220.64   277.1 2222.46   319.4 2223.95   355.6 2223.26
   429.6 2224.09   491.4 2222.54   503.4 2222.59     527 2223.52   537.9 2224.55
   542.8 2225.69   553.1 2228.96   566.8 2234.18   587.2 2246.56   625.3 2265.58
#Mann= 6 ,-1,0
       0     .05       0     120     .06       0   194.3    .045       0
   227.4     .06       0     270     .05       0  563.31      .1       0
Bank Sta=194.3,227.4
XS Rating Curve= 0 ,0
Exp/Cntr(USF)=0,0
Exp/Cntr=0.3,0.1

Type RM Length L Ch R = 1 ,1495    ,150.2,156.2,160.9
XS GIS Cut Line= 2
2187432.32845763411809.1771570012187063.90042716411298.401932937
#Sta/Elev= 30
       0  2231.1    39.5 2229.52   126.2 2222.53   198.6 2221.72   202.2 2221.23
   209.3 2218.65   223.6 2218.27   226.9 2216.62   237.9 2207.61   243.7 2203.68
   252.3 2201.43   266.9 2202.49   271.3 2204.88   274.5 2207.82   281.1  2212.7
   287.4  2216.2   295.9 2218.77   310.7 2221.32   394.6 2220.99   429.9 2222.61
     470 2226.98   493.2 2229.67   503.1 2232.09   521.6 2238.38   552.4 2250.01
   567.2 2256.48   578.9 2262.85   588.3 2270.08   591.8 2271.83   629.8 2286.35
#Mann= 6 ,-1,0
       0     .05       0     110     .06       0     230     .05       0
   237.9    .045       0   274.5     .05       0     470      .1       0
Bank Sta=237.9,274.5
XS Rating Curve= 0 ,0
Exp/Cntr(USF)=0,0
Exp/Cntr=0.3,0.1

Type RM Length L Ch R = 1 ,1338    ,174.1,178.5,175.5
XS GIS Cut Line= 4
2187485.11372864411760.8165039042187457.64490696411622.455031733
2187379.30789698411436.2774625612187234.84224222411268.412441177
#Sta/Elev= 30
       0 2229.95      73 2223.75     140 2220.58   177.2 2219.89   181.5 2218.99
   186.1 2216.93   203.2  2216.2   207.3 2213.89   217.22207.198   224.9  2201.6
   229.2 2199.02   233.6 2198.56   242.3  2200.2   250.1 2204.01   255.3 2207.31
   259.6 2211.23   268.6 2216.75   272.6 2218.41     277 2219.48   286.7 2220.96
   335.6 2223.17   375.8  2224.1     446 2223.24     458 2223.75   470.5 2225.08
   482.8 2227.07   494.2 2229.94   513.4 2235.15   531.8 2241.47   564.5 2248.14
#Mann= 5 ,-1,0
       0     .05       0     140     .06       0   217.2    .045       0
   255.3     .05       0  543.05      .1       0
Bank Sta=217.2,255.3
XS Rating Curve= 0 ,0
Exp/Cntr(USF)=0,0
Exp/Cntr=0.3,0.1

Type RM Length L Ch R = 1 ,1160    ,100.6,201,227.8
BEGIN DESCRIPTION:
xs 4
END DESCRIPTION:
XS GIS Cut Line= 4
2187537.47513226411739.2267120432187603.40030429411534.126176825
2187564.94395394411436.1540461632187321.38706837411246.619176564
#Sta/Elev= 30
       0 2229.97   107.2 2225.08   157.6 2222.02   174.4 2222.17     187 2216.56
   216.5 2217.03   220.7  2216.4     231 2212.84   242.2 2206.98   249.5 2202.97
   264.9 2198.58   268.1 2198.64   272.3 2200.77   276.6 2204.39   282.1 2206.81
   293.8 2211.91   302.4 2214.95   311.2 2217.26   320.5 2218.71   331.9 2218.97
   367.3 2218.02   388.9  2218.6   433.2 2223.78   468.7    2226   524.4 2224.71
   539.6 2225.13   579.5  2228.6   602.7  2229.2   619.8  2231.2   629.3 2233.23
#Mann= 5 ,-1,0
       0     .05       0  225.44     .06       0   242.2    .045       0
   282.1     .06       0  330.68     .05       0
Bank Sta=242.2,282.1
XS Rating Curve= 0 ,0
Exp/Cntr(USF)=0,0
Exp/Cntr=0.5,0.2

Type RM Length L Ch R = 1 ,959     ,138.8,117.6,114.1
BEGIN DESCRIPTION:
xs 3
END DESCRIPTION:
XS GIS Cut Line= 6
2187543.97331535411740.7946816482187608.78391938 411550.75821247
2187635.63857807411517.7058918242187647.09083524411494.646673752
2187750.47715485411494.502869111 2187981.0975016 411509.87875475
#Sta/Elev= 30
       0 2230.14   109.5 2225.15   160.2 2222.21   177.1 2222.16   181.3 2221.26
   185.5 2218.51   189.8 2216.83     194 2216.49   207.2 2216.86   223.4 2218.31
   231.5 2217.65   252.9 2212.78   282.2 2209.89   298.2 2205.36   308.8 2200.18
   318.2  2198.8   322.2  2197.5   326.2  2197.4   332.22200.205   338.2 2204.27
   346.2 2212.57   350.2 2214.83   367.5 2220.08   386.2 2222.68   398.3 2223.59
   434.3  2224.2   472.9 2223.89   551.9 2228.16   578.7 2228.33   603.6 2229.73
#Mann= 5 ,-1,0
       0     .05       0   231.5     .06       0   308.8    .045       0
   332.2     .06       0   472.9     .05       0
#XS Ineff= 2 , 0
           230.8 2216.86   408.2         2218.58
Permanent Ineff=
       F       F
Bank Sta=308.8,332.2
XS Rating Curve= 0 ,0
Exp/Cntr(USF)=0,0
Exp/Cntr=0.5,0.3

Type RM Length L Ch R = 1 ,841     ,185.5,181.4,171
BEGIN DESCRIPTION:
xs 2
END DESCRIPTION:
XS GIS Cut Line= 6
2187557.00807401411745.1389730342187635.68183751411575.870078164
2187704.91346696411572.1446880732187753.62087711 411586.65066483
2187844.39106688411562.1762851782187977.89190655411557.932488949
#Sta/Elev= 30
       0  2230.4    48.5 2228.23    88.2 2225.92   105.8  2225.3   145.5 2222.68
   163.2 2222.33     172 2221.77   180.8 2221.59   207.2 2221.94   231.5 2222.79
   235.2 2222.48   243.2 2219.57   250.5 2218.56   259.4 2218.28   280.3 2218.86
   292.8 2218.37     297 2217.22   305.3 2212.78   309.5 2210.86   313.4 2209.94
   321.9 2208.78   334.3 2210.02   359.2 2213.92   373.9 2216.76   388.4 2220.49
   400.6 2222.32   416.1 2222.98   488.7 2227.59   508.7 2227.11   534.4 2227.15
#Mann= 4 ,-1,0
       0     .05       0  305.99     .06       0   313.4    .045       0
   334.3     .06       0
#XS Ineff= 2 , 0
           304.6  2216.5   341.7            2218
Permanent Ineff=
       F       F
Bank Sta=313.4,334.3
XS Rating Curve= 0 ,0
Exp/Cntr(USF)=0,0
Exp/Cntr=0.5,0.3

Type RM Length L Ch R = 1 ,660     ,206.2,199.2,188.3
XS GIS Cut Line= 3
2187718.09003105411849.3271515422187929.70169437411673.323220031
2187974.46570007411585.829936158
#Sta/Elev= 30
       0 2229.62    75.4 2223.19     112 2221.04   127.6 2220.65   132.8 2219.81
     138 2217.74   140.8 2217.19   153.6 2216.65   162.9 2214.85   169.2 2213.16
   184.8 2206.61     189 2205.77   194.7 2205.61   214.6 2206.82   220.3 2206.47
   226.4 2205.38   231.7 2205.81     2332206.391   236.8 2208.43     243 2213.31
   247.2 2215.78   251.5 2217.88   257.2 2219.78   262.8 2220.71   284.4 2222.26
   306.9 2223.28   315.8 2224.31   347.3 2226.16   360.8 2226.52   373.5 2226.02
#Mann= 5 ,-1,0
       0     .05       0     170      .1       0   220.3    .045       0
     233      .1       0  335.24     .06       0
Bank Sta=220.3,233
XS Rating Curve= 0 ,0
Exp/Cntr(USF)=0,0
Exp/Cntr=0.3,0.1

Type RM Length L Ch R = 1 ,461     ,237.8,238.6,211.7
XS GIS Cut Line= 4
2188014.01875422411954.1654345322188054.49073744411779.831762977
2188036.63440211411712.618420312 2188017.7639215411613.717578279
#Sta/Elev= 30
       0 2227.91    25.7 2225.73    62.6 2223.69    70.8 2221.69    82.6 2219.54
    91.4 2217.21    99.6 2213.65   105.9 2211.39   120.1 2206.77   132.4 2203.19
   140.6  2200.1     141 2199.98   144.7 2198.86   145.9 2198.81   157.1 2199.07
   165.3 2199.97   173.5 2200.96   177.6 2201.84   194.1 2209.04   202.4 2210.91
   210.7 2212.16   219.1 2215.09   227.2 2217.36   243.8 2220.36     252 2221.38
   260.2 2221.79   292.7  2221.5     305 2221.79   341.6  2224.2   349.2 2224.68
#Mann= 5 ,-1,0
       0     .05       0   140.6      .1       0     141    .045       0
   165.3      .1       0   341.6     .06       0
Bank Sta=141,165.3
XS Rating Curve= 0 ,0
Exp/Cntr(USF)=0,0
Exp/Cntr=0.3,0.1
